--- NFGAULYRV.prj (project) ---

Proj Title=NFGAULYRV
Current Plan=p01
Default Exp/Contr=0,0
English Units
Geom File=g01
Flow File=f01
Plan File=p01
Background Map Layer=Inundation Boundary (01pct Value_0)
Y Axis Title=Elevation
X Axis Title(PF)=Main Channel Distance
X Axis Title(XS)=Station
BEGIN DESCRIPTION:
----------MODEL BY WOOD PLC 2021----------
Stream Name: North Fork Gauley River
Flood Zone: Approximate
Pocahontas County, WV
HEC-RAS Version: RAS 6.1
Vertical Datum: NAVD88
Projection: NAD 1983 StatePlane West Virginia S FIPS 4702 (US Feet)
Terrain: 1-meter LIDAR (FEMA Region III 3DEP collected 2016-2018)
Land Use: 2019 NLCD
Hydrologic Method:
WV 2010 Regional Regression Equations
Model Notes:
Model extends beyond county boundary on the downstream end
END DESCRIPTION:
DSS Export Rating Curves= 0
DSS Export Rating Curve Sorted= 0
DSS Export Volume Flow Curves= 0
DXF OffsetX= 0
DXF OffsetY= 0
DXF ScaleX= 0
DXF ScaleY= 0

--- NFGAULYRV.p01 (plan) ---

Plan Title=Floodplain
Program Version=6.10
Short Identifier=Floodplain
Geom File=g01
Flow File=f01
Subcritical Flow
K Sum by GR= 0
Std Step Tol= 0.01
Critical Tol= 0.01
Num of Std Step Trials= 20
Max Error Tol= 0.3
Flow Tol Ratio= 0.001
Split Flow NTrial= 30
Split Flow Tol= 0.02
Split Flow Ratio= 0.02
Log Output Level= 0
Friction Slope Method= 1
Unsteady Friction Slope Method= 2
Unsteady Bridges Friction Slope Method= 1
Parabolic Critical Depth
Global Vel Dist= 0 , 0 , 0
Global Log Level= 0
CheckData=True
Encroach Param=-1 ,0,0, 0
Mapping Interval=1HOUR
Computation Time Step Use Courant=        0
Computation Time Step Use Time Series=    0
Computation Time Step Count To Double=0
Computation Time Step Max Doubling=0
Computation Time Step Max Halving=0
Computation Time Step Residence Courant=0
Run HTab= 0
Run UNet= 0
Run Sediment= 0
Run PostProcess= 0
Run WQNet= 0
Run RASMapper=-1
UNET Theta= 0
UNET Theta Warmup= 0
UNET ZTol= 0
UNET ZSATol= 0
UNET MxIter= 0
UNET Max Iter WO Improvement= 0
UNET MaxInSteps= 0
UNET DtIC= 0
UNET DtMin= 0
UNET MaxCRTS= 0
UNET WFStab= 0
UNET SFStab= 0
UNET WFX= 1
UNET SFX= 1
UNET Gravity=32.174
UNET 1D Methodology=Finite Difference
UNET DSS MLevel= 1
UNET Pardiso=0
UNET DZMax Abort= 0
UNET Use Existing IB Tables= 0
UNET Froude Reduction=False
UNET Froude Limit= 0
UNET Froude Power= 0
UNET D1 Cores= 0
UNET WindReference=Eulerian
UNET WindDragFormulation=Hsu (1988)
UNET D2 Coriolis=0
UNET D2 Cores= 0
UNET D2 Theta= 1
UNET D2 Theta Warmup= 1
UNET D2 Z Tol= 0.01
UNET D2 Volume Tol= 0.01
UNET D2 Max Iterations= 20
UNET D2 Equation= 0
UNET D2 RampUpFraction=0.1
UNET D2 TimeSlices= 1
UNET D2 Turbulence Formulation=Non-Conservative (original)
UNET D2 Eddy Viscosity=0.3
UNET D2 Transverse Eddy Viscosity=0.1
UNET D2 Smagorinsky Mixing=0
UNET D2 BCVolumeCheck=0
UNET D2 Cores=0
UNET D2 SolverType=PARDISO (Direct)
UNET D2 Minimum Iterations= 2147483647
UNET D2 Maximum Iterations= 2147483647
UNET D2 Restart Number= 10
UNET D2 Relaxation Coeff=1.3
UNET D2 SOR Precondition Iterations= 10
UNET D2 ILUT Maximum Fill= 8
UNET D2 ILUT Tolerance=1E-08
UNET D1D2 MaxIter= 0
UNET D1D2 ZTol=0.01
UNET D1D2 QTol=0.1
UNET D1D2 MinQTol=1
Write IC File= 0
Write IC File at Fixed DateTime=0
Write IC File at Sim End=0
Echo Input=False
Echo Parameters=False
Echo Output=False
Write Detailed= 0
HDF Write Warmup=0
HDF Write Time Slices=0
HDF Flush=0
HDF Compression= 1
HDF Chunk Size= 1
HDF Spatial Parts= 1
HDF Use Max Rows=0
HDF Fixed Rows= 1
Calibration Method= 0
Calibration Iterations= 20
Calibration Max Change=0.05
Calibration Tolerance=0.2
Calibration Maximum=1.5
Calibration Minimum=0.5
Calibration Optimization Method= 1
WQ AD Non Conservative
WQ ULTIMATE=-1
WQ Max Comp Step=1HOUR
WQ Output Interval=15MIN
WQ Output Selected Increments= 0
WQ Output face flow=0
WQ Output face velocity=0
WQ Output face area=0
WQ Output face dispersion=0
WQ Output cell volume=0
WQ Output cell surface area=0
WQ Output cell continuity=0
WQ Output cumulative cell continuity=0
WQ Output face conc=0
WQ Output face dconc_dx=0
WQ Output face courant=0
WQ Output face peclet=0
WQ Output face adv mass=0
WQ Output face disp mass=0
WQ Output cell mass=0
WQ Output cell source sink temp=0
WQ Output nsm pathways=0
WQ Output nsm derived pathways=0
WQ Create Restart=0
WQ Fixed Restart=0
WQ System Summary=0
WQ Write To DSS=0
Sorting and Armoring Iterations= 10
XS Update Threshold= 0.02
Bed Roughness Predictor= 0
Hydraulics Update Threshold= 0.02
Energy Slope Method= 1
Volume Change Method= 1
Sediment Retention Method= 0
Sediment TS Multiplier= 1
Warm Up Method= 0
XS Weighting Method= 0
Number of US Weighted Cross Sections= 1
Number of DS Weighted Cross Sections= 1
Upstream XS Weight=0
Main XS Weight=1
Downstream XS Weight=0
Number of DS XS's Weighted with US Boundary= 1
Upstream Boundary Weight= 1
Weight of XSs Associated with US Boundary= 0
Number of US XS's Weighted with DS Boundary= 1
Downstream Boundary Weight= 0.5
Weight of XSs Associated with DS Boundary= 0.5
Percentile Method= 0
Sediment Output Level= 3
Mass or Volume Output= 0
Output Increment Type= 1
Profile and TS Output Increment= 1
Transport Output Increment 1
XS Output Flag= 0
XS Output Increment= 10
Read HDF5 Sediment Hotstart= 0
Sediment Hotstart Type= 0
Write Gradation File= 0
Read Gradation Hotstart= 0
Write HDF5 File= 1
Write Binary Output= 1
Write DSS Sediment File= 0
DSS Sediment Output Type= 1
SV Curve= 0
Specific Gage Flag= 0
Subcell Erosion Methods= 0
Subcell Deposition Methods= 0
Advection Scheme= 1
Matrix Solver= 0
Implicit Weighting Factor= 1
Maximum Outer Loop Convergence Iterations= 5
Convergence Maximum Absolute= 0.001
Convergence RMSE= 0.0001
Grain Fractions Max Abs Error= 0.001
Max Subgrid Regions= 1
Max Subgrid Length Scale= 3.402823E+38
Initial Layer Thickness= 3.402823E+38
Min Layer Thickness= 3.402823E+38
Max Layer Thickness= 3.402823E+38
Number of Layers= 5

--- NFGAULYRV.f01 (steady flow) ---

Flow Title=Flow
Program Version=6.10
Number of Profiles= 6
Profile Names=01pct,10pct,04pct,02pct,0_2pct,01plus
River Rch & RM=NFGAULYRV,Main            ,8367
     717     382     506     609     998    1060
River Rch & RM=NFGAULYRV,Main            ,4957
     803     430     568     682    1110    1190
River Rch & RM=NFGAULYRV,Main            ,1716
    1060     572     752     900    1460    1560
River Rch & RM=NFGAULYRV,Main            ,1244
    1220     662     868    1037    1676    1800
Boundary for River Rch & Prof#=NFGAULYRV,Main            , 1
Up Type= 0
Dn Type= 1
Dn Known WS=3176.3
Boundary for River Rch & Prof#=NFGAULYRV,Main            , 2
Up Type= 0
Dn Type= 1
Dn Known WS=3175.4
Boundary for River Rch & Prof#=NFGAULYRV,Main            , 3
Up Type= 0
Dn Type= 1
Dn Known WS=3175.8
Boundary for River Rch & Prof#=NFGAULYRV,Main            , 4
Up Type= 0
Dn Type= 1
Dn Known WS=3176.1
Boundary for River Rch & Prof#=NFGAULYRV,Main            , 5
Up Type= 0
Dn Type= 1
Dn Known WS=3177.1
Boundary for River Rch & Prof#=NFGAULYRV,Main            , 6
Up Type= 0
Dn Type= 1
Dn Known WS=3177.3
DSS Import GetInterval= 0
DSS Import GetPeak= 0
DSS Import FillOption= 0

--- NFGAULYRV.g01 (geometry) ---

Geom Title=Geometry
Program Version=6.10

River Reach=NFGAULYRV       ,Main
Reach XY= 30
     2202612.583      514447.554     2202116.887      514349.536
     2200822.272      514220.426      2200553.09      514278.566
     2200500.203      514389.368     2200342.797      514456.507
     2200236.804        514456.8     2200087.266      514362.854
     2199889.531      514356.392     2199824.764      514381.661
     2199710.069      514531.062     2199540.569      514477.382
     2199416.403       514574.45     2198806.534      514557.057
     2198726.688      514612.564     2198778.587      514725.111
     2198755.431      514758.401     2198608.813      514808.823
     2198170.437      514857.877     2197924.164       515119.22
     2197563.073       515107.12     2197509.704      515202.254
     2197419.683      515232.834      2197356.08      515315.999
     2196784.808      515650.783     2196284.556      515803.594
     2196033.504      515989.637     2195793.879      516056.283
     2195431.574      516089.669     2195299.202      516236.131

Type RM Length L Ch R = 1 ,8367    ,66.3,72.4,81.8
XS GIS Cut Line= 4
2202591.16018061514268.3852773832202597.56196266 514420.96108289
2202614.63338145514499.916394831 2202680.7851293514648.224345638
#Sta/Elev= 30
       0 3368.15     8.8 3368.84    12.8 3369.82    16.8 3369.86    20.8  3367.4
    24.8 3364.13    28.8 3363.25    36.8 3364.66    44.8 3360.96    48.8 3359.89
    64.9 3363.82    80.9 3362.39    88.9  3361.1   108.9 3360.37   158.5 3363.57
   165.2 3362.44   169.3  3359.4   173.4 3355.13   176.33353.793   181.6 3352.85
   188.7 3353.04  192.643353.791   202.2 3357.23     248 3357.88   256.8  3358.9
   268.9 3359.15   287.4 3361.04   335.5 3362.12   374.7 3364.08395.8823 3366.04
#Mann= 3 ,-1,0
       0      .1       0   176.3    .045       0  192.64      .1       0
Bank Sta=176.3,192.64
XS Rating Curve= 0 ,0
Exp/Cntr(USF)=0,0
Exp/Cntr=0.3,0.1

Type RM Length L Ch R = 1 ,8294    ,120.5,121.2,122.9
XS GIS Cut Line= 4
2202576.22268916514260.9165316592202542.07985156 514418.82715554
2202515.40575969514515.9208499542202484.46381312 514635.42078154
#Sta/Elev= 30
       0 3368.16    16.6 3367.52    28.9 3368.31      33  3367.8    40.6  3364.6
    57.6 3359.58    65.7 3360.16      81 3358.05    98.5  3356.9   139.4 3356.54
   151.7 3355.16   176.4 3357.44   180.6  3356.7   184.7 3353.64  190.07 3350.66
   197.2  3349.8   209.6 3349.94  215.28 3350.66   217.9 3351.28   222.1 3354.49
   226.2 3358.46   230.4 3359.76   238.7 3359.17   249.6 3356.93   255.3 3356.87
   267.7 3358.62   275.9 3360.69   282.3 3361.27   313.1 3361.82   385.7 3368.62
#Mann= 3 ,-1,0
       0      .1       0  190.07    .045       0  215.28      .1       0
Bank Sta=190.07,215.28
XS Rating Curve= 0 ,0
Exp/Cntr(USF)=0,0
Exp/Cntr=0.3,0.1

Type RM Length L Ch R = 1 ,8173    ,149.5,149.1,147.9
XS GIS Cut Line= 4
2202465.53288275514238.3244174132202433.00846041514368.422106774
2202396.87021337514480.4506726132202355.31122926514610.548361974
#Sta/Elev= 30
       0 3364.25    11.2 3363.68    19.4 3364.11    35.9 3363.12    48.3 3363.86
    56.5 3361.73    64.8 3355.42    68.9    3354    81.3 3354.42   134.9 3353.41
   147.5 3352.27   160.1 3353.69     164 3353.43  171.173348.034   172.7 3347.14
   179.9    3347  187.963348.034   202.1    3353   214.8 3354.34   224.3 3356.61
   235.8 3355.92   244.2 3356.39   249.8 3355.34     282 3352.72   315.6 3352.83
     324 3355.23   336.6 3361.65   349.2 3365.43   357.6  3365.5   388.4 3369.49
#Mann= 3 ,-1,0
       0      .1       0  171.17    .045       0  187.96      .1       0
Bank Sta=171.17,187.96
XS Rating Curve= 0 ,0
Exp/Cntr(USF)=0,0
Exp/Cntr=0.3,0.1

Type RM Length L Ch R = 1 ,8024    ,165.2,164.1,163.2
XS GIS Cut Line= 4
2202320.97989457514202.0746325692202286.64855988514330.365409578
 2202259.5448746 514436.973238362202228.82736461514576.105489482
#Sta/Elev= 30
       0 3360.96    11.5 3356.41    23.9  3350.7    35.9 3350.37      57 3350.97
    69.5 3349.98     115 3350.08     144 3348.33   148.1 3348.45   160.5 3350.17
   164.6 3349.36   168.7 3346.72  175.523344.125   181.1  3343.2   185.2 3343.16
  193.523344.127   201.7  3346.9     210 3348.29   226.5 3350.43   247.1 3351.86
   259.7 3351.42   275.8 3349.58     284 3349.81   292.2 3351.09   304.5 3349.34
   345.4 3349.58   353.2 3350.02   357.7 3351.71     370  3358.6   385.3 3363.86
#Mann= 3 ,-1,0
       0      .1       0  175.52    .045       0  193.52      .1       0
Bank Sta=175.52,193.52
XS Rating Curve= 0 ,0
Exp/Cntr(USF)=0,0
Exp/Cntr=0.3,0.1

Type RM Length L Ch R = 1 ,7860    ,172.1,171,168.5
XS GIS Cut Line= 4
2202152.93704581514109.9221026052202124.02644818514285.192600772
2202098.72967525514429.7455889512202078.85363937514554.422541255
#Sta/Elev= 30
       0 3358.62    13.9 3352.01    19.5 3350.49    84.4 3350.06    92.5 3351.01
   104.7 3350.66   112.8 3349.94   124.9 3346.08   128.8 3345.44   177.6 3344.84
   189.8 3343.95   210.1 3343.97   226.4 3345.91  235.243340.234   238.5 3339.35
   254.8 3339.44  259.393340.235     267 3343.77   279.1 3345.97   299.4 3344.29
   308.8 3346.47   331.9  3346.7   344.1 3347.51   372.4 3347.46   388.6 3346.53
   408.9 3347.11     417 3349.61   429.1 3357.19   437.2  3363.6   450.6 3368.95
#Mann= 5 ,-1,0
       0      .1       0  177.64     .08       0  235.24    .045       0
  259.39     .08       0  277.64      .1       0
Bank Sta=235.24,259.39
XS Rating Curve= 0 ,0
Exp/Cntr(USF)=0,0
Exp/Cntr=0.3,0.1

Type RM Length L Ch R = 1 ,7689    ,194.8,195.7,196.9
XS GIS Cut Line= 4
2201974.05272294514068.3631185032201946.94903766514285.192600772
 2201937.9144759 514404.448816022201923.45917708514539.967242437
#Sta/Elev= 30
       0 3356.88     4.9 3356.12    16.9  3356.5      21  3354.9      29 3348.19
    33.1 3345.84    37.1 3345.39    97.6 3343.99   198.3 3343.76   218.5 3340.15
   246.6 3341.63   258.6 3343.38   262.6 3342.11  269.383337.004   270.7 3336.32
   282.7 3336.01  288.113337.007   294.7 3340.53   326.8 3345.09   334.8 3344.05
   342.9 3345.65   354.9    3344   375.1 3344.91   399.2 3343.25   407.2 3341.72
   419.3 3342.12   423.3 3343.42   438.5 3355.58   443.4  3358.7   474.4  3372.6
#Mann= 5 ,-1,0
       0      .1       0  218.52     .08       0  269.38    .045       0
  288.11     .08       0  318.52      .1       0
#XS Ineff= 2 , 0
          258.53 3343.42
Permanent Ineff=
       T       F
Bank Sta=269.38,288.11
XS Rating Curve= 0 ,0
Exp/Cntr(USF)=0,0
Exp/Cntr=0.3,0.1

Type RM Length L Ch R = 1 ,7493    ,311.6,310.8,310.1
XS GIS Cut Line= 4
2201773.48545184514099.0806284912201757.22324067514274.351126659
2201742.76794186514375.5382183842201726.50573069514512.863557154
#Sta/Elev= 30
       0 3356.85    42.3 3350.99    54.3  3348.3   109.7 3338.44   118.6  3338.2
   130.7  3336.7   166.8 3336.58   178.9 3335.37     191 3335.46   203.1 3333.54
  206.473332.068   211.2 3330.51   215.2 3331.15  217.453332.066   243.5 3342.79
   251.6 3343.97   263.7 3344.61   279.9 3342.81   283.9 3341.53     292 3337.42
     296 3336.36     300 3336.07   320.2 3337.09   343.3 3340.44   348.4 3341.93
   384.6 3358.19   388.6 3360.31   400.7 3368.78   408.1 3371.86   416.5  3374.6
#Mann= 5 ,-1,0
       0      .1       0  196.02     .08       0  206.47    .045       0
  217.45     .08       0  388.24      .1       0
#XS Ineff= 2 , 0
                          264.03          3344.7
Permanent Ineff=
       F       F
Bank Sta=206.47,217.45
XS Rating Curve= 0 ,0
Exp/Cntr(USF)=0,0
Exp/Cntr=0.3,0.1

Type RM Length L Ch R = 1 ,7183    ,254.3,255.2,256.3
XS GIS Cut Line= 4
2201460.88961491514091.8529790832201446.43431609 514243.63361667
2201439.20666668514370.1174813272201431.97901727514480.339134814
#Sta/Elev= 30
       0 3359.61    25.4 3352.79    37.5 3348.45    53.6 3345.61    82.6 3338.86
    93.6 3336.88   101.8 3332.37   109.8 3329.95   117.9 3329.25   186.1 3328.72
   190.1 3328.12  197.733324.039   202.1 3323.18   218.1 3323.33  222.523324.039
   231.9 3327.49   238.2 3330.45   242.2 3332.99   246.2 3335.99   250.2 3339.94
   254.6 3345.39   258.4 3348.64     266 3350.02   288.7 3351.91   314.3 3355.65
   322.1 3355.74     330 3356.85   350.4 3361.62   370.4 3367.74   389.6 3372.31
#Mann= 3 ,-1,0
       0      .1       0  197.73    .045       0  222.52      .1       0
Bank Sta=197.73,222.52
XS Rating Curve= 0 ,0
Exp/Cntr(USF)=0,0
Exp/Cntr=0.3,0.1

Type RM Length L Ch R = 1 ,6927    ,214.5,214.8,214.7
XS GIS Cut Line= 4
2201218.76335971514064.7492937992201198.88732383514198.460807865
2201186.23893737514319.5239354642201168.16981384514455.042361882
#Sta/Elev= 30
       0 3358.71    12.6 3351.21    30.8 3343.23    62.5 3334.18    73.2 3332.18
    85.4 3332.72    89.4  3332.2    97.5 3329.44   101.5  3329.4   113.7 3325.06
   116.2 3324.79   158.3 3324.31   166.1 3323.73   178.1 3318.61  182.123317.767
   193.6 3316.89  202.883317.768   206.3  3319.1   214.3 3320.61   230.4 3330.57
   234.4 3331.58   238.4 3330.84   242.5 3330.92   290.9 3337.38     307 3334.98
   339.3 3336.26   343.3 3336.84   355.4 3340.78     367 3343.37   393.6 3348.08
#Mann= 5 ,-1,0
       0      .1       0  182.12    .045       0  202.88      .1       0
  225.18     .08       0   326.9      .1       0
Bank Sta=182.12,202.88
XS Rating Curve= 0 ,0
Exp/Cntr(USF)=0,0
Exp/Cntr=0.3,0.1

Type RM Length L Ch R = 1 ,6713    ,216.5,210.2,205.8
XS GIS Cut Line= 4
2201005.54770214514032.2248714592200985.67166627514180.391684342
2200971.21636745514310.4893737032200958.56798099514431.552501303
#Sta/Elev= 30
       0 3337.32       9 3334.09    17.1 3329.68    21.1 3328.42    29.2 3326.61
    41.3 3325.68    77.6 3319.62    81.7  3319.2    89.8 3320.33   109.9 3320.66
   162.4 3319.41   176.9 3316.87  185.213312.693   194.6 3311.47   198.7 3311.48
  203.483312.693   214.7 3320.16   222.7 3323.82   234.7 3324.91   242.9 3324.11
     259 3329.77   274.7  3329.9   291.1 3331.33   299.2 3331.02   311.2 3327.08
   339.4 3327.12   363.5 3330.62   379.6 3336.09   387.7 3337.12   402.1 3341.35
#Mann= 5 ,-1,0
       0      .1       0  159.49     .08       0  185.21    .045       0
  203.48     .08       0  360.39      .1       0
Bank Sta=185.21,203.48
XS Rating Curve= 0 ,0
Exp/Cntr(USF)=0,0
Exp/Cntr=0.3,0.1

Type RM Length L Ch R = 1 ,6502    ,162.9,163.3,164.3
XS GIS Cut Line= 4
2200752.57997283513988.8589750052200758.00070989514160.515648468
2200788.71821988514312.2962860562200814.01499281514409.869553076
#Sta/Elev= 30
       0 3328.87    12.3 3324.42    32.3 3319.94    84.4    3320    96.4 3317.63
   100.4 3317.41   156.4 3316.09   188.7 3313.46   205.1 3314.04   213.2 3311.96
   221.7 3313.01   225.1 3312.18  229.113310.087   233.6 3309.21     250 3309.19
     254 3309.22  258.513310.088   266.3 3311.42   282.6 3311.12   286.7 3311.72
   294.9  3317.2     303 3323.65   307.1  3324.3   315.3 3324.57   331.6 3323.17
   348.2 3324.43   364.7 3327.01   377.1 3328.02   389.5 3331.25   427.4 3335.42
#Mann= 5 ,-1,0
       0      .1       0     100     .08       0  201.74      .1       0
  229.11    .045       0  258.51      .1       0
#XS Ineff= 2 , 0
          221.12 3313.64
Permanent Ineff=
       F       F
Bank Sta=229.11,258.51
XS Rating Curve= 0 ,0
Exp/Cntr(USF)=0,0
Exp/Cntr=0.3,0.1

Type RM Length L Ch R = 1 ,6339    ,205.5,202.3,196.9
XS GIS Cut Line= 4
2200593.57168583 514024.997222052200604.41315995514198.460807865
2200626.09610817514353.8552701572200660.42744287514464.076923643
#Sta/Elev= 30
       0  3324.1     8.2 3323.25    40.3 3316.27    48.3 3316.95    60.3 3315.29
    92.4 3314.08   104.4 3314.78   132.4  3313.9   168.5  3309.9   176.5 3311.26
   204.8 3311.93   208.9 3311.32   216.9 3307.01     225  3306.6   233.1 3308.33
   238.3  3307.2   245.2 3305.86   258.9 3306.97   269.4  3307.9   281.6 3306.06
   297.7 3308.35   321.9  3308.9   338.4 3312.67   356.9 3326.76   363.5 3330.32
   371.9 3330.81   388.6 3329.91     418 3332.98   434.7 3336.84   446.1 3337.24
#Mann= 3 ,-1,0
       0      .1       0   238.3    .045       0   258.9      .1       0
Bank Sta=238.3,258.9
XS Rating Curve= 0 ,0
Exp/Cntr(USF)=0,0
Exp/Cntr=0.3,0.1

Type RM Length L Ch R = 1 ,6137    ,107.4,110.2,113.6
XS GIS Cut Line= 4
2200429.14266178514046.6801702772200463.47399647514333.979234282
2200505.03298057514431.5525013032200542.97813997514509.249732449
#Sta/Elev= 30
       0 3325.34      23 3322.16    30.2 3319.57    34.7 3316.74    38.8 3315.78
    50.9 3314.48    54.9 3315.09    83.1 3313.23    95.2 3311.23   127.4 3309.94
   163.7 3305.14   183.8  3309.1   192.1 3309.43     208 3308.45   220.1 3305.04
   231.7 3304.23   314.6 3307.98   321.8  3307.2   331.9 3303.82   347.93302.313
   359.4 3301.11  368.243302.313   375.4 3305.28   392.8 3307.69   397.2 3309.63
   406.1  3314.7   419.5 3325.65   423.9 3327.52   448.1 3332.13   481.9 3340.63
#Mann= 3 ,-1,0
       0      .1       0   347.9    .045       0  368.24      .1       0
#XS Ineff= 2 , 0
          314.08 3308.18
Permanent Ineff=
       F       F
Bank Sta=347.9,368.24
XS Rating Curve= 0 ,0
Exp/Cntr(USF)=0,0
Exp/Cntr=0.3,0.1

Type RM Length L Ch R = 1 ,6027    ,273.5,284.5,297.5
XS GIS Cut Line= 4
2200297.23806007514044.8732579242200380.35602827514400.834991315
2200407.45971355514500.2151706882200425.52883708514552.615628903
#Sta/Elev= 30
       0 3322.47    16.7 3320.99    57.8 3310.16    61.9  3309.3    70.1 3309.27
    78.4 3307.74     140 3307.14   159.2 3304.29   176.9 3305.23   189.3 3301.91
   209.8 3303.21   230.3 3302.56   259.1 3305.03   271.4 3304.22   283.7 3306.11
     292  3306.6   337.1 3304.56   345.4 3305.28   353.6 3304.61   372.2 3304.87
   386.6 3304.09   394.8 3302.19  398.983300.519   415.6 3299.41  428.623300.521
   432.2  3301.8   440.9 3308.07   457.1 3322.02   461.3 3323.62     524 3336.39
#Mann= 3 ,-1,0
       0      .1       0  398.98    .045       0  428.62      .1       0
#XS Ineff= 2 , 0
          292.41 3306.73
Permanent Ineff=
       F       F
Bank Sta=398.98,428.62
XS Rating Curve= 0 ,0
Exp/Cntr(USF)=0,0
Exp/Cntr=0.3,0.1

Type RM Length L Ch R = 1 ,5742    ,224.9,217.9,210.7
XS GIS Cut Line= 4
2200138.22977307514048.4870826292200152.68507189514337.593058987
2200098.47770132514482.1460471662200111.12608779514545.387979494
#Sta/Elev= 30
       0 3311.47     4.7 3309.99    36.7    3306    72.8 3306.12    76.8 3305.87
    84.8  3303.7   120.8 3302.35   128.9 3302.79   148.9 3301.07   176.9 3300.15
   209.5 3300.66     217 3299.99     229 3296.85     245 3296.88   289.5 3300.05
   310.4  3300.7   314.7 3300.04  323.513294.946   331.7 3294.19  351.043294.948
   367.2 3297.16   387.3 3298.66   408.6 3297.68   429.4 3298.64   438.5 3305.24
   446.9 3308.37   463.3 3317.23   487.7 3321.82   495.9 3324.72   508.3 3327.02
#Mann= 3 ,-1,0
       0      .1       0  323.51    .045       0  351.04     .08       0
#XS Ineff= 2 , 0
          310.23 3300.97  387.46         3299.21
Permanent Ineff=
       F       F
Bank Sta=323.51,351.04
XS Rating Curve= 0 ,0
Exp/Cntr(USF)=0,0
Exp/Cntr=0.3,0.1

Type RM Length L Ch R = 1 ,5524    ,117.4,106.6,95.1
XS GIS Cut Line= 4
2199906.94499198514061.135469095 2199917.7864661514254.475090784
2199925.01411551514402.6419036672199930.43485256514523.705031267
#Sta/Elev= 30
       0 3312.59       5 3310.27    16.1 3301.99    20.1 3299.72    27.8 3297.13
    40.1 3294.87    80.9 3294.96   108.2 3296.79   124.2 3297.01   144.3 3296.48
   156.3 3295.38   176.3 3295.35   192.3 3294.26   200.4 3294.62   216.4 3292.96
   244.5  3292.6   260.4 3294.33   276.4 3292.52   284.5 3292.57  288.733291.525
   296.5 3289.71   300.5 3289.94  306.243291.526   312.5 3293.38   332.5 3295.83
   340.5  3298.8   360.5  3302.3   404.9  3308.7   433.6 3312.01   463.2 3318.71
#Mann= 5 ,-1,0
       0      .1       0  233.64     .08       0  288.73    .045       0
  306.24     .08       0  323.64      .1       0
#XS Ineff= 2 , 0
          260.18 3295.34
Permanent Ineff=
       F       F
Bank Sta=288.73,306.24
XS Rating Curve= 0 ,0
Exp/Cntr(USF)=0,0
Exp/Cntr=0.3,0.1

Type RM Length L Ch R = 1 ,5417    ,100.6,97.5,94.1
XS GIS Cut Line= 4
2199738.30088432514090.2664827922199776.30025109514335.296882304
2199900.78093533514462.3982125332199908.64287328514565.913728904
#Sta/Elev= 30
       0    3314     4.2 3312.36    15.1 3305.55    35.3  3294.9    39.4 3294.06
    43.4 3294.36    51.5 3292.42   189.1 3292.25   201.3 3292.71   221.6 3291.38
   245.8 3293.06   254.9    3292   302.9 3291.91   306.6 3291.21   312.2 3288.84
   319.9 3288.12   331.2 3288.84     357 3292.75   373.5  3297.8   379.4  3298.4
   390.7 3296.54   421.7  3305.1   448.7 3310.84   456.7 3311.35   472.8 3315.69
   484.8 3317.73   492.8 3319.94   504.9 3321.64   516.9 3321.42   529.7 3323.71
#Mann= 4 ,-1,0
       0      .1       0     200     .08       0   312.2    .045       0
   331.2      .1       0
#XS Ineff= 2 , 0
          245.07 3294.48
Permanent Ineff=
       F       F
Bank Sta=312.2,331.2
XS Rating Curve= 0 ,0
Exp/Cntr(USF)=0,0
Exp/Cntr=0.3,0.1

Type RM Length L Ch R = 1 ,5320    ,186.2,205.3,220.6
XS GIS Cut Line= 4
2199653.96480121514106.9425664432199702.53024372514418.144588578
2199818.99882937514498.7254026072199845.06759002514596.670021273
#Sta/Elev= 30
       0 3319.43    10.4 3317.56    17.9 3314.22    34.7 3303.21    50.8 3294.34
      67  3292.5   164.2 3292.49   176.3 3291.44   208.7 3291.01   263.9 3288.58
   321.8 3288.93   336.4 3287.78   352.8 3288.51   365.6 3290.02   370.5 3289.85
   378.7 3287.68   390.2 3287.16   407.23287.788   418.7 3289.21   428.8 3292.18
   436.2  3292.8     442  3294.4   447.7 3297.82   459.1 3306.94   463.3 3309.45
   467.4 3310.85   475.9  3312.9   496.4 3315.68   524.9  3323.1     558 3330.28
#Mann= 5 ,-1,0
       0      .1       0     180     .08       0     280      .1       0
   378.7    .045       0   407.2      .1       0
#XS Ineff= 2 , 0
          300.88 3293.06
Permanent Ineff=
       F       F
Bank Sta=378.7,407.2
XS Rating Curve= 0 ,0
Exp/Cntr(USF)=0,0
Exp/Cntr=0.3,0.1

Type RM Length L Ch R = 1 ,5115    ,164,158.2,149.2
XS GIS Cut Line= 4
2199565.43855741 514162.322560822199606.99754151514455.042361882
2199608.80445386514527.3188559722199626.87357739514588.753875948
#Sta/Elev= 30
       0 3305.31      15 3292.25    22.6  3288.8    27.1 3288.29    35.2 3289.08
    67.5    3290    83.7 3288.27    91.8 3289.25   107.5 3289.38   124.1 3287.54
   136.2 3287.98   144.3 3286.74   152.4 3288.94   160.6 3289.36   233.2 3287.04
   277.6 3284.13   285.7  3286.5   297.8 3287.17   305.8 3286.71  312.43  3284.3
   313.8 3283.14   329.5 3282.75   333.8 3282.85  339.023284.339   341.8 3285.19
   357.8 3286.78   374.1 3298.07   382.4 3301.75   394.9 3302.79     432 3313.99
#Mann= 3 ,-1,0
       0      .1       0  312.43    .045       0  339.02      .1       0
#XS Ineff= 2 , 0
           256.6 3287.44
Permanent Ineff=
       F       F
Bank Sta=312.43,339.02
XS Rating Curve= 0 ,0
Exp/Cntr(USF)=0,0
Exp/Cntr=0.3,0.1

Type RM Length L Ch R = 1 ,4957    ,210.3,218.3,227
XS GIS Cut Line= 4
2199375.71276043514182.1985966942199458.83072863 514502.02208304
2199494.96897567514572.491664778 2199516.6519239514655.609632981
#Sta/Elev= 30
       0 3298.62    23.7 3285.41    27.9 3284.06    55.3 3287.25    89.9 3285.44
    98.1  3287.2     104 3287.46   118.8 3286.82   122.9 3285.17   127.1 3282.52
   135.3  3285.6   147.7  3286.6   205.6 3284.64   225.9  3283.1   255.2 3284.01
   263.5 3283.29   271.7 3283.97   319.9 3282.83   333.8 3283.55     343 3283.13
  350.453280.243   378.9 3279.16  384.033280.246   401.4 3287.17   418.6 3298.62
   439.3 3308.36   464.8 3317.03     480 3320.62   488.9 3324.01   495.5 3325.66
#Mann= 3 ,-1,0
       0      .1       0  350.45    .045       0  384.03      .1       0
#XS Ineff= 2 , 0
          329.48 3284.36
Permanent Ineff=
       F       F
Bank Sta=350.45,384.03
XS Rating Curve= 0 ,0
Exp/Cntr(USF)=0,0
Exp/Cntr=0.3,0.1

Type RM Length L Ch R = 1 ,4738    ,167.8,170.1,172.2
XS GIS Cut Line= 4
2199216.70447343514297.840987238 2199274.5256687514529.125768324
2199276.33258105514610.4368241752199285.36714281514680.906405912
#Sta/Elev= 30
       0 3293.96    11.7 3291.82    24.1 3286.48    32.3 3284.62    40.5 3284.91
    48.8 3283.72      57 3284.41   127.1 3284.13   164.2 3279.93   168.4 3280.37
   176.6 3282.79   180.4 3283.28   197.2  3283.4   210.1 3281.12   226.1 3280.71
   234.3 3279.71   250.5 3279.52   254.5 3278.38  259.683274.692   262.5 3273.09
   270.5 3272.85   283.1 3273.26  291.413274.692   298.5  3276.8   306.5 3278.28
   314.5 3281.76   330.6 3285.11   366.9 3298.55     379 3301.34   390.8 3307.03
#Mann= 3 ,-1,0
       0      .1       0  259.68    .045       0  291.41      .1       0
Bank Sta=259.68,291.41
XS Rating Curve= 0 ,0
Exp/Cntr(USF)=0,0
Exp/Cntr=0.3,0.1

Type RM Length L Ch R = 1 ,4568    ,213.1,208.7,204.9
XS GIS Cut Line= 4
2199079.37913466514305.068636646 2199115.5173817514464.076923643
2199102.86899524514624.8921229922199122.74503111514713.430828252
#Sta/Elev= 30
       0 3294.19     8.3 3292.95      37 3291.18    61.6 3285.33    70.9 3285.79
    73.9 3285.07      81 3281.09    86.3  3279.6    94.5 3280.88   106.8 3280.33
   110.9 3281.43   119.1 3286.27   123.2  3286.3   131.4 3283.39   147.8 3283.75
     156 3283.06   168.2 3277.92   173.7 3276.66   200.3  3274.4   216.3 3275.89
   232.93272.508   244.4 3271.49  261.973272.507   272.5 3274.82   284.5 3275.02
   308.6 3277.37   332.9 3281.84   353.4 3288.01   373.9 3293.06   415.1 3305.67
#Mann= 3 ,-1,0
       0      .1       0   232.9    .045       0  261.97      .1       0
#XS Ineff= 2 , 0
          216.17 3276.61  276.68         3276.48
Permanent Ineff=
       F       F
Bank Sta=232.9,261.97
XS Rating Curve= 0 ,0
Exp/Cntr(USF)=0,0
Exp/Cntr=0.3,0.1

Type RM Length L Ch R = 1 ,4359    ,210.7,181.2,166.3
XS GIS Cut Line= 3
2198866.16347709514321.330847817 2198907.7224612514592.367700652
2198951.08835765514792.934971751
#Sta/Elev= 30
       0 3283.47    19.2 3280.33    24.1 3278.89    36.3 3273.33    40.3 3272.87
    80.8 3273.28    88.2 3271.76    92.9 3271.66   105.1 3272.63   117.2 3272.38
   137.4 3274.13   157.7 3271.81   165.8 3273.69     182  3274.3   194.1 3272.05
   206.2 3271.98  216.663270.262   222.4 3268.88   229.7 3268.77   238.6 3269.28
  241.013270.262   246.7 3272.05   258.8 3272.89   287.3  3272.8   311.2  3271.4
   377.3 3273.35   401.9 3280.56   426.5  3294.5   442.8 3300.78   479.4 3309.98
#Mann= 3 ,-1,0
       0      .1       0  216.66    .045       0  241.01      .1       0
#XS Ineff= 2 , 0
          181.52 3274.39  283.28         3273.94
Permanent Ineff=
       F       F
Bank Sta=216.66,241.01
XS Rating Curve= 0 ,0
Exp/Cntr(USF)=0,0
Exp/Cntr=0.3,0.1

Type RM Length L Ch R = 1 ,4178    ,266.1,274.1,292.7
XS GIS Cut Line= 4
2198616.80957249514326.7515848732198685.47224187514567.070927721
2198819.18375594 514655.609632982198867.97038945514811.004095273
#Sta/Elev= 30
       0 3277.96    12.3 3275.14    44.1 3270.88   102.4 3270.04   173.4 3269.79
   193.9 3270.33     198 3270.01   206.4 3267.64   210.5 3267.29   227.2    3270
   262.8 3271.12   273.6 3269.05   282.3 3268.41   319.8 3269.05   325.6 3269.87
   344.3 3270.22   358.7 3268.86   368.3 3268.77   382.7 3271.28   425.1 3270.79
   437.9 3269.95   479.4 3270.79   483.2 3271.56   491.6 3276.49   516.8 3288.66
     521 3291.15   537.7 3303.14   547.2 3306.41   562.9 3309.61   573.2 3310.37
#Mann= 3 ,-1,0
       0      .1       0   273.6    .045       0   319.8      .1       0
#XS Ineff= 2 , 0
          262.71 3272.64  382.84         3272.36
Permanent Ineff=
       F       F
Bank Sta=273.6,319.8
XS Rating Curve= 0 ,0
Exp/Cntr(USF)=0,0
Exp/Cntr=0.3,0.1

Type RM Length L Ch R = 1 ,3904    ,186.8,189.1,192.9
XS GIS Cut Line= 4
2198533.69160428 514404.448816022198656.56164424514731.499951774
2198698.12062834 514848.949254672198714.38283951514888.701326419
#Sta/Elev= 30
       0 3284.36     5.1 3282.73    22.1 3274.31    29.8 3272.19    69.1 3270.22
   107.6    3270   120.4  3267.3   136.1  3268.7   151.6 3268.42   167.1 3265.49
   180.2 3269.13   227.2 3269.27   240.1 3267.97   252.9 3269.11   304.2 3268.93
   321.3 3268.04   329.8 3268.46   363.9 3266.49     388 3267.91   393.6 3266.81
  396.78 3264.69   402.1 3263.23   427.5 3263.75   432.1 3264.72   448.7 3276.76
   456.9 3284.71   478.5 3301.12   495.8 3307.47   504.5  3311.8   516.9 3316.66
#Mann= 3 ,-1,0
       0      .1       0  396.78    .045       0   432.1      .1       0
#XS Ineff= 2 , 0
          386.14    3269
Permanent Ineff=
       F       F
Bank Sta=396.78,432.1
XS Rating Curve= 0 ,0
Exp/Cntr(USF)=0,0
Exp/Cntr=0.3,0.1

Type RM Length L Ch R = 1 ,3715    ,240.8,241.4,242.7
XS GIS Cut Line= 4
2198392.75244081514449.621624825 2198468.6427596514717.044652956
2198502.97409429514876.0529399532198517.42939311514942.908696986
#Sta/Elev= 30
       0 3285.75    20.3    3284    34.8 3279.23    49.4 3275.53   109.3 3268.82
   136.8 3263.94     170 3265.43   190.8  3264.2     200 3265.31   232.3 3264.38
   286.3 3265.24   298.6 3262.78   321.5  3261.6   339.5 3264.64   351.8 3263.53
   364.1 3263.65  373.76 3261.23   376.3 3260.38   388.6 3259.81   396.8 3260.01
     404 3261.19   409.1 3262.79   417.3  3267.6   427.4 3274.82   433.6  3280.2
   437.7 3282.49   449.3 3284.25   466.4 3285.39   482.7 3288.12   509.1  3295.3
#Mann= 3 ,-1,0
       0      .1       0  373.76    .045       0     404      .1       0
#XS Ineff= 2 , 0
          341.91 3265.57
Permanent Ineff=
       F       F
Bank Sta=373.76,404
XS Rating Curve= 0 ,0
Exp/Cntr(USF)=0,0
Exp/Cntr=0.3,0.1

Type RM Length L Ch R = 1 ,3474    ,211.9,199.5,189.2
XS GIS Cut Line= 4
 2198184.9575203514520.0912065632198233.74415381514751.375987649
2198262.65475145514906.7704499412198295.17917379514989.888418144
#Sta/Elev= 30
       0 3289.98      35 3286.89    74.7  3279.9   111.5  3275.7   127.8 3272.65
   156.5 3270.47     181 3267.47   189.2 3265.75   201.4 3262.03   238.2 3261.21
   242.3 3260.18   246.3 3258.09   253.7 3257.17     283 3259.11   311.4 3259.14
   315.5 3258.69  321.943256.419   331.8 3255.21   339.9 3255.54   344.23256.418
   348.1 3257.34   360.3 3265.52   363.5  3267.1   370.4 3270.07   376.5 3271.84
   405.6 3272.79   420.6 3274.85   437.6  3276.3   474.3 3281.81   483.7 3283.93
#Mann= 3 ,-1,0
       0      .1       0  321.94    .045       0   344.2      .1       0
#XS Ineff= 2 , 0
          305.83 3261.36
Permanent Ineff=
       F       F
Bank Sta=321.94,344.2
XS Rating Curve= 0 ,0
Exp/Cntr(USF)=0,0
Exp/Cntr=0.3,0.1

Type RM Length L Ch R = 1 ,3274    ,184,186.2,189.4
XS GIS Cut Line= 4
2197957.28656392514642.9612465152198049.43909388514899.542800532
 2198139.7847115514989.888418144 2198184.9575203515073.006386347
#Sta/Elev= 30
       0 3287.15    22.8 3283.87    35.3 3281.33    41.5 3279.23    53.4 3276.99
    66.1 3271.16    83.1 3260.36    87.4  3258.5    91.6 3257.56   168.1 3257.34
     201 3258.46   236.1 3258.09   248.9 3259.32   257.4 3258.59   280.6 3259.57
   293.5 3258.44  303.843254.558   310.4 3253.28   333.1 3253.57  338.153254.556
   354.9 3256.83   374.7 3256.38   378.3 3257.81   389.6  3265.7   397.3 3269.69
   413.2 3273.72   422.4 3273.38   444.4 3279.38     485 3288.39     495 3291.63
#Mann= 3 ,-1,0
       0      .1       0  303.84    .045       0  338.15      .1       0
#XS Ineff= 2 , 0
          281.63  3260.3  356.44         3259.32
Permanent Ineff=
       F       F
Bank Sta=303.84,338.15
XS Rating Curve= 0 ,0
Exp/Cntr(USF)=0,0
Exp/Cntr=0.3,0.1

Type RM Length L Ch R = 1 ,3088    ,242.6,249.8,256
XS GIS Cut Line= 4
2197791.05062751 514679.099493562197946.44508981515033.254314598
2198006.07319743515138.0552310282198029.56305801515176.000390425
#Sta/Elev= 30
       0  3291.7    37.2  3282.3    72.3 3264.29    89.6 3254.08      94  3252.8
   120.2 3252.79   129.9 3254.43   150.8 3253.87   159.5 3255.12     177  3255.5
   194.5 3253.95   255.6 3255.89   273.1 3254.28   290.9 3255.52     308 3255.37
   347.4 3252.17   360.5 3253.04   375.9 3256.41   386.7  3255.9   395.9  3254.1
   418.9 3254.17   431.6 3252.09   446.5 3250.94   451.1 3252.09   467.2 3258.23
   478.7 3266.57   483.3 3268.86   502.4 3271.99     514 3275.07     552 3289.46
#Mann= 3 ,-1,0
       0      .1       0   431.6    .045       0   451.1      .1       0
#XS Ineff= 2 , 0
          377.56 3256.52
Permanent Ineff=
       F       F
Bank Sta=431.6,451.1
XS Rating Curve= 0 ,0
Exp/Cntr(USF)=0,0
Exp/Cntr=0.3,0.1

Type RM Length L Ch R = 1 ,2838    ,217.2,208.8,201.4
XS GIS Cut Line= 4
2197601.32483053514839.9146929092197733.22943224515053.130350473
  2197742.263994515181.4211274812197814.54048809515315.132641547
#Sta/Elev= 30
       0 3282.74    14.6 3279.85      32 3269.51    43.7 3264.15    58.6 3255.06
    67.3  3250.7      72 3249.92   110.5 3249.18     125 3250.45   151.2 3250.77
   194.8 3249.83   217.9 3252.47   227.3 3252.12   236.7  3252.9   254.8 3251.94
   266.8 3248.43   286.9 3248.74   294.9 3250.38   302.9 3249.73   309.7 3248.06
     327 3246.75   332.2 3247.77     343 3250.07     359  3257.1   367.1 3256.93
   392.7 3259.54   433.7 3266.13   465.4 3272.71   525.2 3282.92   531.3 3284.96
#Mann= 3 ,-1,0
       0      .1       0   309.7    .045       0   332.2      .1       0
#XS Ineff= 2 , 0
          237.62 3252.88
Permanent Ineff=
       F       F
Bank Sta=309.7,332.2
XS Rating Curve= 0 ,0
Exp/Cntr(USF)=0,0
Exp/Cntr=0.3,0.1

Type RM Length L Ch R = 1 ,2629    ,258.6,258,255.4
XS GIS Cut Line= 4
2197451.35110529514980.8538563832197520.01377468515094.689334574
2197590.48335642515199.4902510042197707.93265931515358.498538001
#Sta/Elev= 30
       0 3277.16     9.6 3276.02    21.2 3272.59    42.4 3269.36    51.8  3266.5
      79 3261.64    89.1 3261.72    99.9 3257.88   108.6 3252.01   117.2 3248.83
   146.4 3247.33   152.1 3246.24   164.9 3244.82   175.2 3245.96   195.4 3246.97
   224.2 3245.88   235.7 3247.44   256.4 3247.23   270.2 3249.06   276.2 3247.55
     316 3246.13   327.4 3248.39   353.2 3248.85   376.5 3253.56   401.8 3255.98
   410.2 3259.77   416.9 3265.44   435.4  3275.5   447.6 3280.79   456.9 3283.52
#Mann= 3 ,-1,0
       0      .1       0   152.1    .045       0   175.2      .1       0
#XS Ineff= 2 , 0
          132.01    3250
Permanent Ineff=
       F       F
Bank Sta=152.1,175.2
XS Rating Curve= 0 ,0
Exp/Cntr(USF)=0,0
Exp/Cntr=0.3,0.1

Type RM Length L Ch R = 1 ,2371    ,279.3,281.4,282.1
XS GIS Cut Line= 4
2197261.62530831515114.5653704492197353.77783827515262.732183332
2197440.50963118515369.3400121142197503.75156351515459.685629726
#Sta/Elev= 30
       0 3266.06    36.1 3256.96    42.7 3254.04    59.6 3248.21    73.7 3241.45
    78.4 3240.95    97.3  3242.5   111.2 3239.55   120.8 3238.73     135 3239.35
   144.4 3242.22   166.4 3244.59     191 3243.59   200.7 3240.87   206.4 3240.32
  218.01 3240.92   226.3 3241.93   234.8 3244.39   249.8 3245.74   260.4 3245.94
     267 3245.26   275.6 3242.09   285.9 3240.53   306.6 3243.07   326.4 3244.22
   331.7 3245.66   346.2 3251.41   380.5 3268.28   399.6 3271.37   422.2 3277.77
#Mann= 3 ,-1,0
       0      .1       0   200.7    .045       0  218.01      .1       0
Bank Sta=200.7,218.01
XS Rating Curve= 0 ,0
Exp/Cntr(USF)=0,0
Exp/Cntr=0.3,0.1

Type RM Length L Ch R = 1 ,2090    ,89.9,89.4,89.2
XS GIS Cut Line= 4
2197023.11287781515242.8561474572197115.26540778515394.636785045
2197173.08660305515486.7893150092197283.30825654515654.832163768
#Sta/Elev= 30
       0  3262.8    30.8 3258.79    54.2 3250.86    71.4 3247.89    89.8 3240.29
   110.2 3234.21   117.7 3233.64   140.8 3235.34   148.5 3238.04   157.1 3239.83
   177.6 3238.99   185.3 3239.45   197.5 3238.24   224.4 3238.17   232.5  3240.1
   252.6 3241.71   256.1 3241.53   261.3 3239.94   289.2 3241.02   313.1 3239.81
   322.7 3241.09   351.4 3237.67   370.5 3236.84   375.3 3238.03   380.1 3240.98
     404  3257.9   413.6 3261.47   437.8 3263.79   466.5  3263.4487.3216 3266.57
#Mann= 3 ,-1,0
       0      .1       0   197.5    .045       0   224.4      .1       0
Bank Sta=197.5,224.4
XS Rating Curve= 0 ,0
Exp/Cntr(USF)=0,0
Exp/Cntr=0.3,0.1

Type RM Length L Ch R = 1 ,2001    ,101.3,100.3,99.7
XS GIS Cut Line= 4
2196950.65842599515297.9090167842197042.86516332515447.196115327
2197124.82670762515575.9928277952197178.97987082515671.126763141
#Sta/Elev= 30
       0 3263.32    29.6 3255.23    74.4 3238.49    93.6 3237.53   102.6 3235.06
   109.5 3234.03   126.1 3233.29   135.5 3232.03   144.9 3232.39   154.3 3236.75
     192 3237.89   196.8 3237.13   198.1 3236.35   201.5 3235.07   212.6 3236.22
   222.6 3237.76   230.1 3236.79   239.5 3233.83   253.7  3233.9   282.1 3237.68
   291.6 3237.38   305.8 3238.26   338.7 3243.79   357.9 3245.34   375.5 3248.07
   380.1 3247.96   401.8 3251.42   407.7 3250.81   426.2  3253.3   437.6 3253.75
#Mann= 3 ,-1,0
       0      .1       0   198.1    .045       0   212.6      .1       0
#XS Ineff= 2 , 0
          153.49 3242.13
Permanent Ineff=
       F       F
Bank Sta=198.1,212.6
XS Rating Curve= 0 ,0
Exp/Cntr(USF)=0,0
Exp/Cntr=0.3,0.1

Type RM Length L Ch R = 1 ,1900    ,182.1,184.3,187.2
XS GIS Cut Line= 4
2196873.13915258515345.8501515352196959.87094548515497.630789123
2197010.46449135515571.7141955652197108.03775837515709.039534335
#Sta/Elev= 30
       0 3263.21    25.2 3258.91    36.1 3255.94    42.8 3253.27    77.5 3235.23
    86.8 3232.72     119 3231.72   130.7 3233.49   155.9 3233.14   179.1 3235.42
     184 3234.33   188.8 3231.64   198.5 3230.57   209.2  3231.6     213 3232.54
   217.9 3237.17   222.7  3239.1   240.9 3240.86   249.5 3242.69   266.3 3243.24
   285.9 3246.33   295.1    3247   310.5 3247.65   324.2 3246.51   336.5 3248.72
   375.8 3250.02   384.9 3251.75   408.6 3252.39   421.7 3255.05432.9846    3255
#Mann= 3 ,-1,0
       0      .1       0   188.8    .045       0   209.2      .1       0
#XS Ineff= 2 , 0
          178.22 3237.69
Permanent Ineff=
       F       F
Bank Sta=188.8,209.2
XS Rating Curve= 0 ,0
Exp/Cntr(USF)=0,0
Exp/Cntr=0.3,0.1

Type RM Length L Ch R = 1 ,1716    ,158.1,160.7,163.4
XS GIS Cut Line= 4
2196732.48580554515460.7434964572196801.63924124 515583.43507593
2196870.79267694515708.3574113942196899.79250482515837.741258839
#Sta/Elev= 30
       0 3265.92    55.9  3258.3    78.6 3256.61    94.1 3254.41   101.5 3251.94
   111.7 3246.45   120.5 3241.44   133.7 3232.69   138.2 3231.73   147.4 3232.46
   164.6 3231.87   170.3 3228.85   173.4 3226.01   175.53224.927   199.9 3224.18
   206.8 3224.92   211.4 3227.16     216 3230.71   220.4 3232.97   236.9 3232.36
   245.2 3232.75   270.8 3244.85   279.4 3247.53   298.7 3251.78   313.2 3254.41
   317.3    3254   333.7 3254.95   365.8 3260.06   382.8 3261.53   416.2 3268.23
#Mann= 3 ,0,0
       0      .1       0   175.5    .045       0   206.8      .1       0
Bank Sta=175.5,206.8
XS Rating Curve= 0 ,0
Exp/Cntr(USF)=0,0
Exp/Cntr=0.3,0.1

Type RM Length L Ch R = 1 ,1555    ,306.8,311.2,314.3
XS GIS Cut Line= 4
2196614.75068621515537.3828608722196656.30967031515634.956127893
2196715.93777793515783.1229407762196748.46220027515871.661646036
#Sta/Elev= 30
       0 3260.79      78 3252.25    86.7 3248.77   104.1 3232.34   112.8 3227.19
   121.4    3229   126.1 3228.48   138.6 3230.07   142.9 3229.39   151.6 3223.55
  155.133222.026   177.4 3221.06  182.753222.026   190.4 3225.07   193.7 3225.59
     206 3225.02   220.6 3225.79   229.2  3227.6   237.8 3234.87   246.4 3240.71
   255.2 3248.29   263.7 3254.23     285 3261.54   293.5 3265.55   302.1 3267.47
   320.5 3275.52   327.6 3276.98   340.4 3277.56   348.9 3281.35360.0938 3282.94
#Mann= 3 ,-1,0
       0      .1       0  155.13    .045       0  182.75      .1       0
#XS Ineff= 2 , 0
                          195.38         3228.59
Permanent Ineff=
       F       F
Bank Sta=155.13,182.75
XS Rating Curve= 0 ,0
Exp/Cntr(USF)=0,0
Exp/Cntr=0.3,0.1

Type RM Length L Ch R = 1 ,1244    ,237.5,232.8,227.7
XS GIS Cut Line= 4
2196332.87235926515587.9764067352196374.43134336515730.722482561
2196399.72811629515848.1717854572196428.63871393515952.972701887
#Sta/Elev= 30
       0 3268.14    13.3 3264.58      23 3261.28    38.7 3251.02    51.2 3240.27
    55.4 3237.36    76.2    3226    80.4  3224.4    88.7 3222.54   101.2 3221.62
   158.9 3222.35   167.6 3220.47  176.213216.265   204.4 3215.33   212.6 3215.47
  214.643216.263   216.7 3217.08   224.8  3227.7   228.9 3231.56   249.4 3247.22
   253.5 3249.33   257.6 3250.16   265.8 3250.46     283 3252.73   294.8 3255.68
   307.2 3257.04   331.8 3261.76   340.4 3264.22   369.4 3269.73377.5309 3271.93
#Mann= 3 ,-1,0
       0      .1       0  176.21    .045       0  214.64      .1       0
Bank Sta=176.21,214.64
XS Rating Curve= 0 ,0
Exp/Cntr(USF)=0,0
Exp/Cntr=0.3,0.1

Type RM Length L Ch R = 1 ,1011    ,240.6,241.8,243.2
XS GIS Cut Line= 4
2196110.62213993515700.004972573 2196161.2156858515833.716486639
2196220.84379342515960.2003512962196262.40277752516045.125231851
#Sta/Elev= 30
       0 3272.69    26.9 3263.78    61.1 3258.01    78.2 3256.49    91.1 3254.03
    95.7 3251.74   103.9 3245.03   116.7 3235.61   125.3 3229.89   138.1 3223.16
   146.8 3217.64   160.1 3217.08   165.8 3217.85   168.9 3216.95   177.8 3211.78
  180.023211.313   199.9 3210.55  215.323211.312   235.2 3214.63     244 3218.73
   262.5 3231.04   279.5 3244.71   288.3 3252.86   297.2 3258.31   306.9 3260.86
   324.9 3262.35   332.9 3264.21   350.7 3266.29     364 3269.31 377.346 3271.18
#Mann= 3 ,-1,0
       0      .1       0  180.02    .045       0  215.32      .1       0
Bank Sta=180.02,215.32
XS Rating Curve= 0 ,0
Exp/Cntr(USF)=0,0
Exp/Cntr=0.3,0.1

Type RM Length L Ch R = 1 ,770     ,232.8,238.8,240.8
XS GIS Cut Line= 4
 2195922.7032553515768.6676419582195955.22767764515911.413717785
 2196002.2073988516083.0703912482196025.69725938516160.767622394
#Sta/Elev= 30
       0  3263.6    37.4 3256.51    53.9 3256.25    66.2  3251.9    78.5 3249.81
    91.9 3249.99   119.5 3247.26   131.8 3241.82   148.2 3227.17   173.1 3212.14
   181.2 3209.75   193.9  3209.9     198 3209.07   206.3 3203.36   214.6  3202.1
   222.9 3202.27  228.743200.659   235.3 3199.48  249.313200.659   260.2 3202.75
   264.4 3205.31   269.1 3208.97   280.9 3225.13   285.1 3229.48   314.7 3246.63
   322.4 3249.14   364.2 3257.05   389.3 3264.78   397.6 3268.45405.5443  3269.3
#Mann= 4 ,-1,0
       0     .12       0   196.4      .1       0  228.74    .045       0
  249.31      .1       0
Bank Sta=228.74,249.31
XS Rating Curve= 0 ,0
Exp/Cntr(USF)=0,0
Exp/Cntr=0.3,0.1

Type RM Length L Ch R = 1 ,531     ,246.7,247.1,244.7
XS GIS Cut Line= 4
2195723.94289656515853.5925225142195745.62584478515994.531685988
2195758.27423125516139.0846741672195781.76409183516242.078678245
#Sta/Elev= 30
       0  3240.9    27.9 3237.16      36 3236.87      56 3231.79    72.4 3223.74
      91  3212.2   106.7 3205.13   115.6 3203.88     125 3204.15   137.2 3201.04
   153.3 3200.88   165.3 3199.73   169.3 3198.39   177.4 3192.68  182.433190.903
   205.5 3190.05  217.293190.905   225.6 3193.28   229.6 3196.63   237.6 3208.42
   241.6 3213.39   253.7 3220.29   273.7 3233.94   277.8 3235.81     294 3239.07
   327.8 3243.57   347.3 3248.17   363.7 3249.56   380.1 3253.68393.3413 3258.08
#Mann= 3 ,-1,0
       0      .1       0  182.43    .045       0  217.29      .1       0
Bank Sta=182.43,217.29
XS Rating Curve= 0 ,0
Exp/Cntr(USF)=0,0
Exp/Cntr=0.3,0.1

Type RM Length L Ch R = 1 ,284     ,242.1,234.1,219.6
XS GIS Cut Line= 4
 2195476.3959043515871.6616460362195501.69267723515994.531685988
2195530.60327487516187.8713076772195548.67239839516263.761626471
#Sta/Elev= 30
       0 3245.57     9.7 3239.99    26.1 3237.72    30.1 3235.74    46.5 3225.78
    66.9 3207.77      71 3206.19    83.2 3205.98   103.6 3198.39   111.8 3192.69
   115.9    3191   136.2 3190.51   148.3 3192.65   172.6 3192.07   180.7 3189.59
  192.693182.469     209 3181.54  229.25 3182.47   233.3 3185.03   241.4 3195.07
   245.4 3198.53   269.7 3207.71   277.7 3209.43   292.1 3209.63   302.4 3210.99
   322.3 3216.41   351.1 3229.54   363.2 3231.22     384 3237.31398.9481 3239.48
#Mann= 3 ,-1,0
       0      .1       0  192.69    .045       0  229.25      .1       0
Bank Sta=192.69,229.25
XS Rating Curve= 0 ,0
Exp/Cntr(USF)=0,0
Exp/Cntr=0.3,0.1

Type RM Length L Ch R = 1 ,50      ,,,
XS GIS Cut Line= 4
2195221.62126263516008.9869848062195288.47701967516144.505411224
2195375.20881257516256.5339770632195422.18853373516336.038120561
#Sta/Elev= 30
       0 3244.66     9.1 3240.63      17 3238.31    49.3 3232.14    62.7 3230.37
    79.7  3225.7   105.2 3207.24   116.2 3200.41   138.5 3184.66   148.4 3184.35
   167.1 3188.89   177.3 3185.66   189.8 3185.82   196.4 3182.84   202.7 3176.03
  206.99 3174.09   228.4 3173.11  248.673174.092   255.2 3176.18   263.3 3176.57
   279.7 3183.97   283.5 3186.55   310.4 3209.89   318.3 3215.34   326.1 3217.49
   340.7 3219.35   358.6 3222.96   365.5 3225.49   377.2 3231.83 385.138 3233.91
#Mann= 3 ,-1,0
       0      .1       0  206.99    .045       0  248.67      .1       0
Bank Sta=206.99,248.67
XS Rating Curve= 0 ,0
Exp/Cntr(USF)=0,0
Exp/Cntr=0.3,0.1
LCMann Table=0

Chan Stop Cuts=-1
Use User Specified Reach Order=0
Composite Channel Slope=5
